--- BFKELKRV.prj (project) ---

Proj Title=BFKELKRV
Current Plan=p01
Default Exp/Contr=0,0
English Units
Geom File=g01
Flow File=f01
Plan File=p01
BEGIN DESCRIPTION:
----------MODEL BY WOOD PLC 2022----------
AFH study
Randolph County, WV
HEC-RAS Version: RAS 6.2
Vertical Datum: NAVD88
Projection: NAD 1983 StatePlane West Virginia S FIPS 4702 (US Feet)
Terrain: 1-meter LIDAR (FEMA Region III 3DEP collected 2016-2018)
Land Use: 2019 NLCD
Hydrologic Method:
WV SIR2010-5033 regression equations
Additional Model Notes:
None
END DESCRIPTION:
DSS Export Rating Curves= 0
DSS Export Rating Curve Sorted= 0
DSS Export Volume Flow Curves= 0
DXF OffsetX= 0
DXF OffsetY= 0
DXF ScaleX= 0
DXF ScaleY= 0

--- BFKELKRV.p01 (plan) ---

Plan Title=Floodplain
Program Version=6.20
Short Identifier=Floodplain
Geom File=g01
Flow File=f01
Subcritical Flow
K Sum by GR= 0
Std Step Tol= 0.01
Critical Tol= 0.01
Num of Std Step Trials= 20
Max Error Tol= 0.3
Flow Tol Ratio= 0.001
Split Flow NTrial= 30
Split Flow Tol= 0.02
Split Flow Ratio= 0.02
Log Output Level= 0
Friction Slope Method= 1
Unsteady Friction Slope Method= 2
Unsteady Bridges Friction Slope Method= 1
Parabolic Critical Depth
Global Vel Dist= 0 , 0 , 0
Global Log Level= 0
CheckData=True
Encroach Param=-1 ,0,0, 0
Mapping Interval=1HOUR
Computation Time Step Use Courant=        0
Computation Time Step Use Time Series=    0
Computation Time Step Count To Double=0
Computation Time Step Max Doubling=0
Computation Time Step Max Halving=0
Computation Time Step Residence Courant=0
Run HTab= 0
Run UNet= 0
Run Sediment= 0
Run PostProcess= 0
Run WQNet= 0
Run RASMapper=-1
UNET Theta= 0
UNET Theta Warmup= 0
UNET ZTol= 0
UNET ZSATol= 0
UNET MxIter= 0
UNET Max Iter WO Improvement= 0
UNET MaxInSteps= 0
UNET DtIC= 0
UNET DtMin= 0
UNET MaxCRTS= 0
UNET WFStab= 0
UNET SFStab= 0
UNET WFX= 1
UNET SFX= 1
UNET Gravity=32.174
UNET 1D Methodology=Finite Difference
UNET DSS MLevel= 1
UNET Pardiso=0
UNET DZMax Abort= 0
UNET Use Existing IB Tables= 0
UNET Froude Reduction=False
UNET Froude Limit= 0
UNET Froude Power= 0
UNET D1 Cores= 0
UNET WindReference=Eulerian
UNET WindDragFormulation=Hsu (1988)
UNET D2 Coriolis=0
UNET D2 Cores= 0
UNET D2 Theta= 1
UNET D2 Theta Warmup= 1
UNET D2 Z Tol= 0.01
UNET D2 Volume Tol= 0.01
UNET D2 Max Iterations= 20
UNET D2 Equation= 0
UNET D2 RampUpFraction=0.1
UNET D2 TimeSlices= 1
UNET D2 Turbulence Formulation=Non-Conservative (original)
UNET D2 Eddy Viscosity=0.3
UNET D2 Transverse Eddy Viscosity=0.1
UNET D2 Smagorinsky Mixing=0
UNET D2 BCVolumeCheck=0
UNET D2 Cores=0
UNET D2 SolverType=PARDISO (Direct)
UNET D2 Minimum Iterations= 2147483647
UNET D2 Maximum Iterations= 2147483647
UNET D2 Restart Number= 10
UNET D2 Relaxation Coeff=1.3
UNET D2 SOR Precondition Iterations= 10
UNET D2 ILUT Maximum Fill= 8
UNET D2 ILUT Tolerance=1E-08
UNET D1D2 MaxIter= 0
UNET D1D2 ZTol=0.01
UNET D1D2 QTol=0.1
UNET D1D2 MinQTol=1
Write IC File= 0
Write IC File at Fixed DateTime=0
Write IC File at Sim End=0
Echo Input=False
Echo Parameters=False
Echo Output=False
Write Detailed= 0
HDF Write Warmup=0
HDF Write Time Slices=0
HDF Flush=0
HDF Compression= 1
HDF Chunk Size= 1
HDF Spatial Parts= 1
HDF Use Max Rows=0
HDF Fixed Rows= 1
Calibration Method= 0
Calibration Iterations= 20
Calibration Max Change=0.05
Calibration Tolerance=0.2
Calibration Maximum=1.5
Calibration Minimum=0.5
Calibration Optimization Method= 1
WQ AD Non Conservative
WQ ULTIMATE=-1
WQ Max Comp Step=1HOUR
WQ Output Interval=15MIN
WQ Output Selected Increments= 0
WQ Output face flow=0
WQ Output face velocity=0
WQ Output face area=0
WQ Output face dispersion=0
WQ Output cell volume=0
WQ Output cell surface area=0
WQ Output cell continuity=0
WQ Output cumulative cell continuity=0
WQ Output face conc=0
WQ Output face dconc_dx=0
WQ Output face courant=0
WQ Output face peclet=0
WQ Output face adv mass=0
WQ Output face disp mass=0
WQ Output cell mass=0
WQ Output cell source sink temp=0
WQ Output nsm pathways=0
WQ Output nsm derived pathways=0
WQ Create Restart=0
WQ Fixed Restart=0
WQ System Summary=0
WQ Write To DSS=0
Sorting and Armoring Iterations= 10
XS Update Threshold= 0.02
Bed Roughness Predictor= 0
Hydraulics Update Threshold= 0.02
Energy Slope Method= 1
Volume Change Method= 1
Sediment Retention Method= 0
Sediment TS Multiplier= 1
Warm Up Method= 0
XS Weighting Method= 0
Number of US Weighted Cross Sections= 1
Number of DS Weighted Cross Sections= 1
Upstream XS Weight=0
Main XS Weight=1
Downstream XS Weight=0
Number of DS XS's Weighted with US Boundary= 1
Upstream Boundary Weight= 1
Weight of XSs Associated with US Boundary= 0
Number of US XS's Weighted with DS Boundary= 1
Downstream Boundary Weight= 0.5
Weight of XSs Associated with DS Boundary= 0.5
Percentile Method= 0
Sediment Output Level= 3
Mass or Volume Output= 0
Output Increment Type= 1
Profile and TS Output Increment= 1
Transport Output Increment 1
XS Output Flag= 0
XS Output Increment= 10
Read HDF5 Sediment Hotstart= 0
Sediment Hotstart Type= 0
Write Gradation File= 0
Read Gradation Hotstart= 0
Write HDF5 File= 1
Write Binary Output= 1
Write DSS Sediment File= 0
DSS Sediment Output Type= 1
SV Curve= 0
Specific Gage Flag= 0
Subcell Erosion Methods= 0
Subcell Deposition Methods= 0
Advection Scheme= 1
Matrix Solver= 0
Implicit Weighting Factor= 1
Maximum Outer Loop Convergence Iterations= 5
Convergence Maximum Absolute= 0.001
Convergence RMSE= 0.0001
Grain Fractions Max Abs Error= 0.001
Max Subgrid Regions= 1
Max Subgrid Length Scale= 3.402823E+38
Initial Layer Thickness= 3.402823E+38
Min Layer Thickness= 3.402823E+38
Max Layer Thickness= 3.402823E+38
Number of Layers= 5

--- BFKELKRV.f01 (steady flow) ---

Flow Title=Flow
Program Version=6.20
Number of Profiles= 1
Profile Names=P100yr
River Rch & RM=BFKELKRV,Main,21343
    2210
River Rch & RM=BFKELKRV,Main,11864
    2460
River Rch & RM=BFKELKRV,Main,9012
    2940
Boundary for River Rch & Prof#=BFKELKRV,Main            , 1
Up Type= 0
Dn Type= 3
Dn Slope=0.015927
DSS Import GetInterval= 0
DSS Import GetPeak= 0
DSS Import FillOption= 0

--- BFKELKRV.g01 (geometry) ---

Geom Title=Geometry
Program Version=6.20

River Reach=BFKELKRV        ,Main
Reach XY= 30
     2209599.459      579877.746     2209313.996       579669.27
     2208844.127      578396.498     2208548.217      578248.475
  2208296.842543577866.3721326782208032.69330467577708.352238329
     2207269.001      578190.0562207310.92410406578567.547283092
     2206964.456      578897.8762206631.28476167579086.533304668
     2206076.664      579164.4362205559.86369533579068.652351352
     2204091.878      578077.7512203603.54050369578228.604980344
2203155.06730467578106.912371008     2202364.329      578580.821
     2201256.203      578312.027     2201059.496      578112.821
     2201140.743      577617.569     2201019.579      577155.073
     2200587.072      576870.443      2200329.91      576539.393
     2198634.085      575357.713     2197305.489      575234.658
     2196361.685      574859.0932196363.37305114574552.507031049
2195272.86115233573761.613980344     2194847.151      572994.933
      2194390.09      572753.897     2194061.377      572391.059

Type RM Length L Ch R = 1 ,21343   ,496.3,508.5,520
XS GIS Cut Line= 4
2209834.50056629579690.3947807042209631.40429951579775.637117832
2209405.28231693580054.6196838912209282.18275873580058.022378714
#Sta/Elev= 30
       0 2951.33    28.6 2943.42    58.9 2928.87    79.5 2915.29      98 2910.69
     117 2899.36   129.2 2893.66   162.8 2883.13   180.4 2875.91   203.6 2871.79
   225.4    2862   273.7 2860.45  283.192856.135   289.1 2854.85   301.6 2854.71
  319.382856.132   371.5 2860.41   390.6 2858.59   428.7 2857.82   476.8  2861.2
   511.3 2861.07   525.1 2858.38   556.4 2862.12   574.8  2861.2   580.5 2863.27
   604.5 2878.27   612.5 2884.93   624.5 2897.71   632.5 2903.09   702.5 2927.13
#Mann= 3 ,-1,0
       0      .1       0  283.19    .045       0  319.38      .1       0
Bank Sta=283.19,319.38
XS Rating Curve= 0 ,0
Exp/Cntr=0.3,0.1

Type RM Length L Ch R = 1 ,20834   ,383.8,388.4,394.5
XS GIS Cut Line= 2
2209677.50763339579333.6341669382208980.81628152579613.595050732
#Sta/Elev= 30
       0 2944.64    83.3 2925.49   109.2 2910.79   132.9 2899.47   165.2 2888.91
   188.3 2885.34   199.7 2881.38   252.8 2852.16   280.5 2850.46   303.2 2852.76
   337.7 2851.06   376.5 2852.09   393.7  2847.7   428.1 2848.12  437.022846.556
   477.3 2845.52   487.92846.557   518.7 2862.27   535.8  2874.1   557.5 2891.85
   570.5 2900.02   612.6  2915.9   630.2 2918.27   642.4 2921.79   669.6 2934.48
   680.3 2936.87   721.4 2954.52   734.3 2957.17   742.9 2963.19   750.8 2966.54
#Mann= 3 ,-1,0
       0      .1       0  437.02    .045       0   487.9      .1       0
Bank Sta=437.02,487.9
XS Rating Curve= 0 ,0
Exp/Cntr=0.3,0.1

Type RM Length L Ch R = 1 ,20446   ,416.8,418.4,420.5
XS GIS Cut Line= 2
2209465.19425889579077.200480109 2208887.3175158579172.380178971
#Sta/Elev= 30
       0 2903.26    29.4 2893.26    41.6 2891.39      74 2881.42    90.2 2879.11
   102.4 2875.45   106.4 2873.87   122.6 2862.81   134.8 2856.76     147 2847.97
   155.1 2844.47   219.9 2846.43   232.1 2845.43   248.3 2847.09   276.7 2845.86
   280.8 2845.15  287.992840.455   321.1 2839.07   331.3 2840.43   349.7 2841.87
   406.4 2839.93   414.5 2840.94   430.7 2847.33   459.1 2870.91   479.4    2883
   515.9 2898.61     528  2902.3   540.2 2909.69   552.4 2912.68   585.7 2934.38
#Mann= 3 ,-1,0
       0      .1       0  287.99    .045       0   331.3      .1       0
Bank Sta=287.99,331.3
XS Rating Curve= 0 ,0
Exp/Cntr(USF)=0,0
Exp/Cntr=0.3,0.1

Type RM Length L Ch R = 1 ,20028   ,412.1,395.6,375.7
XS GIS Cut Line= 2
 2209453.8360671578733.9403338752208801.20255017578784.862833606
#Sta/Elev= 30
       0 2931.72     105 2893.12   178.2 2872.49   214.3 2865.05     242 2854.73
   254.4 2848.11   266.5 2847.37   274.5 2845.17   286.5 2839.01   310.6 2834.57
   322.6 2836.66   338.7  2835.7   382.8 2836.76   390.8 2834.99   422.9 2835.89
  434.422832.384   447.4 2831.41  479.752832.383   487.1 2836.12   491.1 2836.79
   511.2 2835.18   515.2 2836.03   521.9 2840.47   543.3 2859.07   571.4 2878.89
   583.4 2883.28   591.5 2891.34   595.5 2893.96   611.5 2903.16   654.6 2920.32
#Mann= 3 ,-1,0
       0      .1       0  434.42    .045       0  479.75      .1       0
#XS Ineff= 2 , 0
          324.48 2846.83
Permanent Ineff=
       F       F
Bank Sta=434.42,479.75
XS Rating Curve= 0 ,0
Exp/Cntr=0.3,0.1

Type RM Length L Ch R = 1 ,19632   ,368.6,369.6,364.7
XS GIS Cut Line= 3
2209069.40108672577992.2203714922209039.72878233578198.907454961
2208697.34256466578586.526219297
#Sta/Elev= 30
       0 2898.26    73.7 2875.79    85.8  2875.1   110.1 2868.04   134.3 2865.31
   175.1 2863.34   182.8 2860.31     203 2848.56   211.8 2846.48   243.9  2844.2
   259.9 2844.99   270.5 2841.25   318.6 2837.44   339.9 2832.77   371.6 2830.97
     400  2832.5     452 2825.85   461.9 2825.73   490.7 2825.11  511.08 2825.76
   521.4 2828.07   548.1 2828.59   558.7 2831.68   600.9 2838.81     613 2845.35
   632.3  2858.2   686.8 2885.65   711.7 2900.52   720.2 2902.54     726 2906.37
#Mann= 3 ,-1,0
       0      .1       0   461.9    .045       0  511.08      .1       0
Bank Sta=461.9,511.08
XS Rating Curve= 0 ,0
Exp/Cntr=0.3,0.1

Type RM Length L Ch R = 1 ,19262   ,441.4,446.2,446.7
XS GIS Cut Line= 2
2208897.24686449 577898.794039612208433.05557904578362.529949268
#Sta/Elev= 30
       0 2906.46    44.9 2892.15    58.1 2890.17    93.9 2879.29   122.2 2867.18
   133.5  2865.7     158 2847.91   182.4 2833.72   190.1 2831.59   212.8 2832.95
   227.7 2820.34   233.3 2819.09   255.9 2821.62   284.2 2820.01   306.8 2821.79
   347.5  2821.2   365.6 2825.67   382.6 2822.61   435.2 2824.81   466.3  2822.4
   473.1 2820.31   501.4 2820.34   512.7 2822.52   524.1 2830.21     537 2849.49
   544.3 2857.53   562.5 2870.81   578.2 2877.25   641.7 2911.46   656.1 2917.42
#Mann= 3 ,-1,0
       0      .1       0   473.1    .045       0   501.4      .1       0
Bank Sta=473.1,501.4
XS Rating Curve= 0 ,0
Exp/Cntr=0.3,0.1

Type RM Length L Ch R = 1 ,18816   ,428,397.3,386.2
XS GIS Cut Line= 4
2208706.98213551577620.9184517082208473.08885337577765.441931903
2208212.67474554577954.0800335452208167.04424878578185.238937464
#Sta/Elev= 30
       0 2945.66    53.8 2924.84    92.6 2905.33   106.7 2899.73   120.9 2896.59
   135.9 2889.67   147.5 2888.52   159.2 2882.74   191.4 2879.29   196.9 2875.66
   208.6 2871.61   229.3 2859.36   252.5 2848.88   276.1 2832.12   310.6 2815.48
   409.4 2814.23   439.1 2810.85   481.6 2810.04  487.87 2810.88   504.6 2816.22
   518.9  2815.4   537.8 2816.93   550.4 2821.56   592.2 2824.58   607.8  2828.9
   632.3 2839.12   688.1 2851.68   742.4  2871.7   783.1 2890.27   832.1 2910.27
#Mann= 3 ,-1,0
       0      .1       0   439.1    .045       0  487.87      .1       0
#XS Ineff= 2 , 0
          406.13 2824.37
Permanent Ineff=
       F       F
Bank Sta=439.1,487.87
XS Rating Curve= 0 ,0
Exp/Cntr=0.3,0.1

Type RM Length L Ch R = 1 ,18419   ,467,450.9,443.6
XS GIS Cut Line= 3
2207966.71423766577390.7013391222207967.92694847 577970.39655335
2207995.74199444578187.945931903
#Sta/Elev= 30
       0 2915.84    46.5 2901.37    87.8 2891.33    90.5 2890.19    98.5 2881.83
   103.7 2878.96   150.5  2876.3   170.5 2865.59   210.5 2836.87   222.5 2826.88
   249.5 2808.96   274.5 2806.24  282.362801.936   310.5 2800.67  324.282801.937
   357.8 2807.17   430.5 2804.67   442.5 2805.52   454.5 2803.65   462.5 2804.74
   502.5 2804.48   526.1 2813.89   570.5 2817.63   594.6 2826.28   614.6  2836.7
   626.9 2839.89     639    2848   671.8 2862.85   691.4 2866.54     799 2907.43
#Mann= 3 ,-1,0
       0      .1       0  282.36    .045       0  324.28      .1       0
#XS Ineff= 2 , 0
                        403.1203            2810
Permanent Ineff=
       F       F
Bank Sta=282.36,324.28
XS Rating Curve= 0 ,0
Exp/Cntr=0.3,0.1

Type RM Length L Ch R = 1 ,17968   ,418.3,410.8,405.8
XS GIS Cut Line= 3
2207393.44111327577637.0827400982207692.58567676578096.849581837
     2207832.441578259.689191805
#Sta/Elev= 30
       0 2899.73    19.2 2891.09    62.2  2876.9    74.3 2874.81      86 2869.54
   103.2 2864.46   107.7 2861.36   114.6 2853.37   122.4 2849.34   138.5 2847.99
   175.5 2848.19   186.2 2846.65     203 2836.33   239.1 2826.53     268 2809.26
   291.2 2799.92  339.872789.513   353.3  2788.2  382.392789.513   396.2 2794.85
   406.8 2796.58   415.7 2795.46   486.9 2794.99   496.4 2792.72   515.5 2794.28
   545.6 2804.35   578.6 2818.69   599.5 2829.92   654.4 2855.39   763.2 2895.25
#Mann= 3 ,-1,0
       0      .1       0  339.87    .045       0  382.39      .1       0
#XS Ineff= 2 , 0
                          487.51          2800.5
Permanent Ineff=
       F       F
Bank Sta=339.87,382.39
XS Rating Curve= 0 ,0
Exp/Cntr=0.3,0.1

Type RM Length L Ch R = 1 ,17557   ,412,405.5,406.7
XS GIS Cut Line= 2
2207149.44613988578102.6227094662207626.80066985 578468.88048683
#Sta/Elev= 30
       0 2848.03    13.5 2845.69    17.3 2843.37    23.7 2837.31    28.6 2835.27
    50.2 2832.64    63.7 2833.24      74 2830.24   104.3 2802.96   114.4 2794.85
   120.7 2784.52   126.4 2780.95   135.6 2779.21   154.7 2778.73   161.9 2780.91
   174.9 2782.56   180.6 2784.67   200.6 2786.67   255.5 2786.13   270.7 2788.26
   321.1 2786.69   336.2 2789.28   376.5  2789.1   396.7 2791.12     432 2812.08
   462.2 2820.16   494.5 2830.97     543 2849.25   563.1 2855.11   601.7  2870.7
#Mann= 3 ,-1,0
       0      .1       0   126.4    .045       0   161.9      .1       0
Bank Sta=126.4,161.9
XS Rating Curve= 0 ,0
Exp/Cntr(USF)=0,0
Exp/Cntr=0.3,0.1

Type RM Length L Ch R = 1 ,17155   ,385.7,386.6,388.8
XS GIS Cut Line= 2
2206937.02059691578338.5133795332207551.58819646578734.675912726
#Sta/Elev= 30
       0 2863.98    56.1 2833.58      65 2831.83    86.1 2816.43   100.9 2813.85
   108.5 2809.21   143.1 2808.83   186.5 2782.53   248.5 2781.06   261.8 2783.12
   270.3 2780.79     275 2780.71   285.5 2782.93   298.8 2779.93   355.9 2779.04
     394 2776.43   408.3 2770.76   423.8 2770.27   441.2 2769.32   456.2 2770.25
   460.6    2774   470.1 2787.95   474.9 2793.09   493.9 2810.38     499 2814.22
     513    2821     551 2845.48   620.6 2873.26   655.7 2889.24   731.2 2914.58
#Mann= 3 ,-1,0
       0      .1       0   423.8    .045       0   456.2      .1       0
Bank Sta=423.8,456.2
XS Rating Curve= 0 ,0
Exp/Cntr=0.3,0.1

Type RM Length L Ch R = 1 ,16771   ,390.4,398.6,412.5
XS GIS Cut Line= 3
2206734.19282488578494.9875649762206841.27507298578675.414706049
2207245.88480751      579033.622
#Sta/Elev= 30
       0  2855.8    11.8 2854.31    23.5 2846.78      63 2828.15    86.3 2819.26
   105.8 2814.26     114 2810.22   129.3 2797.46   165.3 2794.02   193.3 2782.29
   207.7 2774.47   245.7 2772.53   256.4 2774.41   275.5 2773.96   284.9 2776.55
   387.5 2776.52   400.1 2775.77   414.3 2770.26  430.532766.589     471 2765.27
  489.552766.589   507.5 2787.97   526.3 2807.12   550.3  2827.8   582.3 2850.14
     653 2880.14   694.8 2901.26     709 2906.34   725.4 2908.07   750.2 2916.48
#Mann= 3 ,-1,0
       0      .1       0  430.53    .045       0  489.55      .1       0
Bank Sta=430.53,489.55
XS Rating Curve= 0 ,0
Exp/Cntr=0.3,0.1

Type RM Length L Ch R = 1 ,16372   ,377.2,379.1,385.7
XS GIS Cut Line= 3
2206565.75912439578615.4666553172206599.37884984578827.013843102
2206782.65944615579260.458112586
#Sta/Elev= 30
       0 2841.42    17.6 2833.39    54.4 2819.99    62.5 2815.49    78.7    2814
    94.9 2808.59   123.2 2802.74   196.1 2791.49   216.5 2778.25   222.6 2776.08
   234.8 2776.69   259.2    2775   277.9 2772.93   301.9 2767.82   312.1 2767.26
   394.6 2768.48   407.6    2767   439.3 2767.45   461.3 2761.96   490.2 2760.43
  501.852761.962   524.9 2763.73   537.9  2773.3   568.3 2802.32     577 2807.97
   613.3 2823.24   633.5 2835.48   657.9 2853.98   671.2 2857.28   684.8  2871.3
#Mann= 3 ,-1,0
       0      .1       0   461.3    .045       0  501.85      .1       0
Bank Sta=461.3,501.85
XS Rating Curve= 0 ,0
Exp/Cntr=0.3,0.1

Type RM Length L Ch R = 1 ,15993   ,502,511,524.7
XS GIS Cut Line= 2
2206234.76066334578636.1817203632206370.73166171579361.360378354
#Sta/Elev= 30
       0 2871.12    45.8 2853.33    90.5 2830.89   139.4  2813.6   163.1 2800.02
   176.8 2789.94   192.3 2781.56   204.5 2772.28   212.6 2768.82     233 2765.86
   261.5 2765.57   273.7 2764.27   342.9 2766.65   363.2 2763.91   371.4 2764.72
   379.5 2763.81   387.6 2759.11   391.7 2758.45     408 2761.17   433.9 2762.23
  487.732757.132   509.3 2755.73  548.182757.132   550.5  2757.9   566.7 2771.72
   607.4 2791.31   680.7 2815.06   713.2 2829.85   725.4 2838.54   737.8 2841.14
#Mann= 3 ,-1,0
       0      .1       0  487.73    .045       0  548.18      .1       0
#XS Ineff= 2 , 0
        431.8613    2766
Permanent Ineff=
       F       F
Bank Sta=487.73,548.18
XS Rating Curve= 0 ,0
Exp/Cntr(USF)=0,0
Exp/Cntr=0.3,0.1

Type RM Length L Ch R = 1 ,15482   ,388.2,390.5,391.6
XS GIS Cut Line= 2
2205981.63184712578574.1925364882205763.94573417579338.947171503
#Sta/Elev= 30
       0 2896.59    48.9 2881.16      78 2864.93    86.3 2858.22    98.8 2852.57
   127.9 2832.97   148.7 2816.75   173.6  2801.3   194.4 2784.72   227.7 2763.67
   252.6 2751.54   281.8 2753.37   323.3 2750.85   385.2 2752.14   398.2 2754.86
   414.7 2749.88   427.3  2752.5   456.4 2753.33   492.4 2749.13   543.8 2750.96
  554.222748.076   589.4 2746.78  595.122748.075   628.4 2770.38   657.5 2785.81
   719.1 2802.87   755.9 2820.06   768.3  2822.1   776.7 2827.49   795.1 2834.74
#Mann= 3 ,-1,0
       0      .1       0  554.22    .045       0  595.12      .1       0
#XS Ineff= 2 , 0
        437.3022    2757
Permanent Ineff=
       F       F
Bank Sta=554.22,595.12
XS Rating Curve= 0 ,0
Exp/Cntr=0.3,0.1

Type RM Length L Ch R = 1 ,15091   ,387.1,389.8,388.2
XS GIS Cut Line= 2
2205653.70610703578537.3679263422205364.46011421 579263.03383962
#Sta/Elev= 30
       0 2879.62    12.7 2877.79    29.9 2867.92    42.9 2865.25    96.5 2836.04
   133.4 2807.89   146.2 2800.75   176.3 2775.37   202.2 2757.31   236.6 2752.47
   253.9  2745.2   305.5 2744.97   322.8 2741.13     383 2747.02   400.3 2741.75
   443.3 2744.17   457.9 2748.37   464.8 2745.83  470.012740.658   481.3 2738.82
   507.9 2740.62   538.1 2740.67   558.3 2754.81   598.3 2790.75     663 2803.97
   684.5  2812.4   714.6 2829.36   727.5 2829.89   740.4 2838.55   781.2 2849.91
#Mann= 3 ,-1,0
       0      .1       0  470.01    .045       0   507.9      .1       0
#XS Ineff= 2 , 0
        456.8939    2750
Permanent Ineff=
       F       F
Bank Sta=470.01,507.9
XS Rating Curve= 0 ,0
Exp/Cntr=0.3,0.1

Type RM Length L Ch R = 1 ,14702   ,423.5,421.4,422.5
XS GIS Cut Line= 2
2205339.99221239578428.1602141592205003.63099379579079.836337716
#Sta/Elev= 30
       0 2854.13    42.2 2839.58    91.2 2831.16   119.4 2821.93   136.2 2810.85
     155 2794.81   167.7 2785.61   208.4  2750.3   226.2 2739.11   239.7 2736.76
     253 2736.65   338.8 2738.47     348 2735.52  362.252734.369   392.5 2733.08
   412.82734.368   425.2 2738.57   493.5 2736.45   527.8 2738.83   550.3 2750.52
   590.8 2783.79   595.3 2785.08   622.3 2784.91   631.3 2786.62   640.3 2791.29
   649.3 2800.63   653.8 2803.83   667.4 2808.59   698.3 2823.29   733.4  2835.5
#Mann= 3 ,-1,0
       0      .1       0  362.25    .045       0   412.8      .1       0
#XS Ineff= 2 , 0
         299.399    2745  440.94            2745
Permanent Ineff=
       F       F
Bank Sta=362.25,412.8
XS Rating Curve= 0 ,0
Exp/Cntr=0.3,0.1

Type RM Length L Ch R = 1 ,14280   ,399.8,409.6,414.6
XS GIS Cut Line= 2
2204952.74023142 578241.669209172204669.85322848 578831.07294696
#Sta/Elev= 30
       0 2834.74    39.4 2819.05    74.9 2810.62    88.2 2808.74      99 2804.33
   110.4 2804.86   119.3 2801.77   141.4 2787.54   159.2  2779.9   168.1 2774.23
   194.7 2756.38   212.9 2742.67   224.9 2731.84   230.9 2729.04   239.9 2727.59
   257.9 2729.39   269.4 2728.62   296.9 2730.12  313.742727.122   336.7 2725.84
  360.492727.121   374.8 2735.17   390.2 2728.65   437.8 2729.68   447.6 2732.77
   464.7 2732.63   487.5  2741.5   540.8 2770.44   616.2 2792.39   653.8 2805.07
#Mann= 3 ,-1,0
       0      .1       0  313.74    .045       0  360.49      .1       0
#XS Ineff= 2 , 0
                        374.5034            2735
Permanent Ineff=
       F       F
Bank Sta=313.74,360.49
XS Rating Curve= 0 ,0
Exp/Cntr=0.3,0.1

Type RM Length L Ch R = 1 ,13871   ,394.9,386.8,379.5
XS GIS Cut Line= 4
2204633.33841766578113.8320284872204561.12212439578237.294830439
2204352.78846257578453.7092787412204276.56669886578647.727153192
#Sta/Elev= 30
       0 2841.75      78  2786.1   105.8 2771.75   115.1 2764.76   124.4 2760.28
   137.8 2749.64     154 2740.65   160.6 2735.19   171.9 2722.65     179 2719.15
   220.6 2717.99  227.112719.053   236.7 2723.57   242.8 2724.29   292.8 2723.12
     302 2724.88     315 2720.77   324.7 2722.33   348.3 2721.39   386.6 2724.95
   415.2 2722.45     426 2719.07   432.2 2719.03   447.2  2725.2   468.6 2743.53
   474.3 2746.19     503 2752.81   511.6 2757.63   566.9 2777.66   651.9 2805.32
#Mann= 3 ,-1,0
       0      .1       0     179    .045       0  227.11      .1       0
Bank Sta=179,227.11
XS Rating Curve= 0 ,0
Exp/Cntr=0.3,0.1

Type RM Length L Ch R = 1 ,13484   ,412.9,394.3,373.9
XS GIS Cut Line= 3
2204248.80489298577952.8203960962204053.31587005578373.293051413
2204038.18420655578551.114678558
#Sta/Elev= 30
       0 2814.12    15.8    2805    48.9 2782.75    75.4 2769.85    88.6 2756.97
   101.9 2747.22   123.9 2728.72   141.6 2716.36  152.662712.065   172.3 2710.53
   190.1 2710.63  199.172712.065   226.6 2715.51   256.7 2715.84   267.2 2712.78
     318 2713.68     326 2714.73   335.6 2720.36   343.1 2722.03   371.1 2722.52
   397.4 2721.28   419.5 2724.03   445.9 2722.08   458.4 2722.54   475.6 2728.44
   499.7 2742.31   523.7 2753.38   551.9  2757.1   623.7 2789.14   642.2 2796.17
#Mann= 3 ,-1,0
       0      .1       0  152.66    .045       0  199.17      .1       0
Bank Sta=152.66,199.17
XS Rating Curve= 0 ,0
Exp/Cntr=0.3,0.1

Type RM Length L Ch R = 1 ,13090   ,395,411.9,435.5
XS GIS Cut Line= 4
2203769.47287955577872.4332606952203763.35418462 578060.07323845
 2203873.4906933578349.6914649852203873.71731163 578526.22714454
#Sta/Elev= 30
       0 2807.17    24.8 2797.33    44.8 2787.25    56.8 2784.34   128.8 2757.37
   140.8 2749.13   152.8 2747.71   172.5 2737.62   210.3 2712.73   223.2 2709.58
   240.3 2709.16  268.652705.078   283.1 2704.02  325.042705.078   347.3 2709.45
   364.4 2706.36   381.4 2707.42   390.1  2709.8   424.3 2706.98   441.4 2715.53
   479.9  2717.5     490 2722.07   537.1 2749.76   553.1 2752.79   569.1 2760.52
   605.1 2773.16   621.1 2781.12   633.1 2781.98   661.1 2793.29   674.1 2800.27
#Mann= 3 ,-1,0
       0      .1       0  268.65    .045       0  325.04      .1       0
Bank Sta=268.65,325.04
XS Rating Curve= 0 ,0
Exp/Cntr(USF)=0,0
Exp/Cntr=0.3,0.1

Type RM Length L Ch R = 1 ,12678   ,450.1,428.6,386.5
XS GIS Cut Line= 4
2203460.45645171 577875.828373172203459.10040654578070.456756781
2203343.20379965578317.0584253762203362.87980751578497.194107025
#Sta/Elev= 30
       0 2794.15    13.5 2786.15    25.4 2781.23    65.5 2757.87    85.4 2754.75
   121.4 2744.29   137.4 2737.93   173.4 2710.79   189.4 2702.43   206.5 2699.76
   250.7 2700.25  263.462697.455   272.8  2696.2     305 2696.28  309.792697.454
   316.1  2699.5   334.7 2699.15   349.2 2701.07     454 2699.94   479.3 2704.73
   495.4  2712.1   519.5 2728.98   531.6 2735.86   559.8 2744.07   571.9 2749.56
   583.9 2757.54     600 2760.29   616.8 2773.82   632.2  2782.5   648.3 2788.41
#Mann= 3 ,-1,0
       0      .1       0  263.46    .045       0  309.79      .1       0
#XS Ineff= 2 , 0
                          349.43         2707.55
Permanent Ineff=
       F       F
Bank Sta=263.46,309.79
XS Rating Curve= 0 ,0
Exp/Cntr=0.3,0.1

Type RM Length L Ch R = 1 ,12249   ,381.8,385.5,390.6
XS GIS Cut Line= 4
2202923.72239542577996.6664864382202989.73153649578145.341039609
2203173.91990667 578347.651900012203211.12087561 578516.60675122
#Sta/Elev= 30
       0  2790.5     9.3 2786.24    20.8  2783.1    48.7 2765.71    58.3 2758.59
   106.8  2729.1   127.5 2718.14   136.2 2710.12   153.7 2696.49   162.5 2693.84
   184.1  2691.5  197.432687.564   229.4 2686.42  256.79 2687.61   269.1 2690.11
   281.5 2687.11   294.5 2688.03   335.6 2696.52   356.4 2694.87   395.1 2694.89
   413.5 2697.03   424.8 2696.09   452.9 2699.55   461.6 2704.65   486.4  2724.1
   499.3 2730.97   519.7 2746.87   552.5 2765.48     573 2775.79   609.3 2789.91
#Mann= 3 ,-1,0
       0      .1       0  197.43    .045       0  256.79      .1       0
#XS Ineff= 2 , 0
                          269.73         2694.33
Permanent Ineff=
       F       F
Bank Sta=197.43,256.79
XS Rating Curve= 0 ,0
Exp/Cntr=0.3,0.1

Type RM Length L Ch R = 1 ,11864   ,417.9,428.4,441
XS GIS Cut Line= 3
2202613.37098499578141.5494239022202646.02418458578294.586972625
2202871.41727436578640.363411542
#Sta/Elev= 30
       0 2760.76    40.5  2743.1    65.1 2734.83    86.3 2725.44     106 2720.05
   126.4 2705.53   134.6 2702.95     151 2692.61   159.9 2689.55   183.5 2688.49
     197 2685.47   226.3 2682.91   269.4 2682.57  288.722678.691   324.7 2677.27
  339.182678.692   355.3 2684.48   369.7 2684.56   379.2 2687.23   391.2 2695.52
   405.6 2708.27     427 2711.44   434.5 2714.63   446.1 2723.81   455.6 2734.23
   468.1 2742.44   509.7 2754.58   522.5 2760.72   541.6 2764.42   569.2  2778.1
#Mann= 3 ,-1,0
       0      .1       0  288.72    .045       0  339.18      .1       0
Bank Sta=288.72,339.18
XS Rating Curve= 0 ,0
Exp/Cntr=0.3,0.1

Type RM Length L Ch R = 1 ,11435   ,383,386.4,388
XS GIS Cut Line= 2
2202320.53443391578185.0967306442202348.72116456578760.983456282
#Sta/Elev= 30
       0 2752.07     8.1 2751.23    36.1 2738.62    64.2 2729.99   104.2 2712.69
   164.3 2693.12   184.3 2689.58   208.3 2680.15   252.4 2679.82   264.4 2677.57
   280.4 2680.54   288.4 2680.07   304.4 2672.73   328.5 2674.21   336.5 2670.38
   344.5  2668.7   372.5 2672.92   381.5 2670.64   408.6 2669.44   421.6 2670.58
     430 2676.61   444.6 2692.08   472.6 2714.53   500.7 2724.55   512.7 2731.02
   528.7 2732.56   536.7 2737.73   552.7 2744.56   568.8 2746.57   576.6 2751.21
#Mann= 3 ,-1,0
       0      .1       0   381.5    .045       0   421.6      .1       0
Bank Sta=381.5,421.6
XS Rating Curve= 0 ,0
Exp/Cntr=0.3,0.1

Type RM Length L Ch R = 1 ,11049   ,417,419.3,422.5
XS GIS Cut Line= 2
2202018.08166496578137.8448942312201928.13684954578793.157120891
#Sta/Elev= 30
       0 2751.18    39.7 2741.91    55.9 2736.46   108.3 2713.65   116.4 2708.39
   128.5 2704.92     181 2675.79   193.1 2670.48   209.3 2666.88   224.8 2668.94
   249.7 2669.37   261.8  2666.3   314.3 2668.89   318.3 2668.39   337.92660.714
   342.5 2659.52   358.7 2659.38   391.82660.715   411.2 2664.72   431.3 2665.64
   443.5 2668.98   467.7 2681.99   483.9 2688.92   495.9  2692.5   528.2 2698.53
   548.4 2700.35   568.6 2699.15   597.5 2709.36   621.1 2711.94   661.5 2729.34
#Mann= 3 ,-1,0
       0      .1       0   337.9    .045       0   391.8      .1       0
Bank Sta=337.9,391.8
XS Rating Curve= 0 ,0
Exp/Cntr(USF)=0,0
Exp/Cntr=0.3,0.1

Type RM Length L Ch R = 1 ,10629   ,342.4,355.2,364.5
XS GIS Cut Line= 4
2201772.57361849578003.0835660882201606.03197763578217.537680899
2201507.78250807578618.774315477 2201545.9546285578810.127142186
#Sta/Elev= 30
       0 2743.39    46.3 2728.95    58.8 2727.78   119.1 2707.19   176.7 2690.88
   260.9 2674.47   269.7 2668.08   291.7 2665.35   305.8 2656.95   316.5 2656.74
     329 2660.68   350.3 2660.46   382.3 2659.34   398.8 2654.67   411.2 2656.76
   427.6 2663.55  456.242654.855   489.4 2653.33  508.762654.851   518.2 2660.06
   547.3 2658.67   567.7 2668.38   592.4    2671   637.7 2671.11   662.4 2674.56
   691.1 2685.94   727.9 2692.98   817.6  2718.8   829.8 2720.09   879.7 2739.58
#Mann= 3 ,-1,0
       0      .1       0  456.24    .045       0  508.76      .1       0
#XS Ineff= 2 , 0
        425.2083    2665
Permanent Ineff=
       F       F
Bank Sta=456.24,508.76
XS Rating Curve= 0 ,0
Exp/Cntr=0.3,0.1

Type RM Length L Ch R = 1 ,10274   ,396.4,434.4,454.6
XS GIS Cut Line= 4
2201596.31100501577923.5902643512201364.60504678 578101.13272467
2201132.45741154578423.6164239022200974.92902002578504.260072421
#Sta/Elev= 30
       0 2717.99    18.3 2710.65    29.8 2709.07     111  2683.4   146.3 2680.76
   169.6 2674.57   242.1 2663.33   259.1 2657.84   286.5 2654.81   300.8 2650.05
   370.8 2651.48   383.9 2654.48   398.3 2652.16   406.9 2654.43     430 2655.04
   450.1 2648.15   458.5 2649.69   474.3 2656.97  493.342649.886  554.082649.862
   578.8 2654.64   587.7 2658.32   618.9 2657.14     632 2661.94   650.5 2661.27
   684.8 2668.12     759 2691.73   824.4 2717.01   842.4 2720.87   866.2 2730.99
#Mann= 5 ,-1,0
       0      .1       0  491.91     .06       0  493.34    .045       0
  554.08     .06       0  699.26     .08       0
#XS Ineff= 2 , 0
        477.3153    2662
Permanent Ineff=
       F       F
Bank Sta=493.34,554.08
XS Rating Curve= 0 ,0
Exp/Cntr=0.3,0.1

Type RM Length L Ch R = 1 ,9840    ,400.4,393,384.4
XS GIS Cut Line= 4
     2201571.341      577843.4792201337.07091961577954.284046427
2200814.08846394577912.403613483 2200736.1599002577893.986778039
#Sta/Elev= 30
       0 2725.98    30.1 2712.98    69.9 2706.27   127.4 2688.86   145.1 2687.55
   171.6 2678.43     229 2668.52   237.9 2662.98     253 2649.57   260.1 2645.94
   348.3 2647.06     391 2644.86   440.6 2647.32   487.6 2645.98  497.682642.186
   528.9 2640.92  549.412642.194     565 2650.77   581.1 2642.46   601.1 2646.38
   649.3 2646.09   661.3 2648.05   685.4 2646.12   701.5 2640.99   761.7 2644.62
   777.7 2651.93     794    2670   814.7 2684.07   832.6 2699.19   863.9 2719.88
#Mann= 5 ,-1,0
       0      .1       0  497.68    .045       0  549.41      .1       0
  569.15     .06       0  669.15      .1       0
#XS Ineff= 2 , 0
          439.02 2653.64562.3633            2655
Permanent Ineff=
       F       F
Bank Sta=497.68,549.41
XS Rating Curve= 0 ,0
Exp/Cntr=0.3,0.1

Type RM Length L Ch R = 1 ,9447    ,447.1,434.5,423.7
XS GIS Cut Line= 2
2201580.85743391577467.7553815122200685.70943391577633.661381512
#Sta/Elev= 30
       0 2772.87      17 2766.88    33.2 2767.41    65.8 2749.35   155.3 2738.59
   183.8 2733.09   204.1 2726.06   224.4 2723.18     257 2711.98   276.4 2710.14
   293.5 2699.19   366.8 2672.93  420.322633.853   444.1 2632.53  478.832633.852
   492.9 2637.94   509.7  2636.4   521.4 2638.44   530.3 2635.79   561.2 2637.74
   627.2  2635.5   680.1 2645.27   692.3 2642.83   700.4  2645.4   758.1 2645.02
   781.8 2650.42   818.4 2651.31     855  2657.6   875.3 2677.71   910.4 2690.89
#Mann= 5 ,-1,0
       0      .1       0  420.32    .045       0  478.83      .1       0
     560     .06       0     660      .1       0
#XS Ineff= 1 ,-1
 519.195 910.393    2640
Permanent Ineff=
       F
Bank Sta=420.32,478.83
XS Rating Curve= 0 ,0
Exp/Cntr=0.3,0.1

Type RM Length L Ch R = 1 ,9012    ,423.1,409.8,400.5
XS GIS Cut Line= 3
 2201123.5715237576955.7977903992201062.89076302577093.386254341
2200659.52507978577425.808561083
#Sta/Elev= 30
       0 2721.71    27.7 2712.38    36.5 2706.23    67.1 2699.17    71.5 2695.69
   110.8 2678.85   123.9 2676.72   152.2 2666.03   168.9 2654.63   181.5 2637.71
  195.982625.594   219.2 2623.86  238.932625.595   247.2 2628.81   274.3 2627.17
     299 2633.88   319.8 2634.44   368.1 2630.88   402.7 2631.83   413.6 2629.05
   458.2 2632.03   483.4 2629.07   506.4  2629.8     540  2641.4   584.1 2644.31
     604 2648.81   630.8 2661.02   646.3 2664.07   665.8 2680.84   673.1  2683.5
#Mann= 5 ,-1,0
       0      .1       0  195.98    .045       0  238.93      .1       0
  320.38     .06       0  450.38      .1       0
#XS Ineff= 2 , 0
                           333.5         2642.31
Permanent Ineff=
       F       F
Bank Sta=195.98,238.93
XS Rating Curve= 0 ,0
Exp/Cntr=0.3,0.1

Type RM Length L Ch R = 1 ,8603    ,405,424.6,433.1
XS GIS Cut Line= 4
2200913.04536118576641.8239846292200757.01864055576706.070281361
2200589.97826905577113.5753634852200514.71832145577177.821660217
#Sta/Elev= 30
       0 2712.35     8.8 2707.39    18.6 2704.75    44.2 2691.16    58.4 2689.14
    64.5 2686.92    83.1 2675.62   116.6 2662.73   156.4 2639.29   172.1 2633.92
   205.5 2625.54     227 2623.13   325.1 2623.16   340.7 2620.91   353.7 2621.76
  361.892619.514   383.9 2618.31   409.9 2618.32  415.462619.517   422.8 2623.94
   432.4 2624.37   483.4 2621.48   499.8 2624.31     509 2622.48   611.5 2624.76
   616.8 2626.37   637.8 2640.18   651.7 2646.67   664.1 2651.54   708.1 2664.29
#Mann= 6 ,-1,0
       0      .1       0  361.89    .045       0  415.46      .1       0
  468.74     .06       0  488.74      .1       0  578.74     .08       0
#XS Ineff= 2 , 0
          323.48 2629.58435.1539            2630
Permanent Ineff=
       F       F
Bank Sta=361.89,415.46
XS Rating Curve= 0 ,0
Exp/Cntr(USF)=0,0
Exp/Cntr=0.3,0.1

Type RM Length L Ch R = 1 ,8178    ,426.2,405.7,402.3
XS GIS Cut Line= 2
2200686.54084545576374.046142186 2200193.3444713 576764.10494525
#Sta/Elev= 30
       0 2684.13     5.1 2682.59    46.6 2657.84    74.4 2643.53   120.3 2629.48
   129.2 2625.02   145.8 2623.14   157.7 2617.38   172.7 2619.45   220.3 2621.33
   240.3 2617.94   254.5 2617.47   305.8 2620.09   314.3 2619.42  327.07 2613.22
   354.9 2611.95  393.58 2613.22   400.8 2618.16   419.7 2615.11   431.4 2616.14
   456.4 2613.79   482.2 2613.37   497.7 2617.54   507.9 2614.03   527.4 2614.51
   548.7 2625.22   578.9  2656.4   589.5 2664.68     619 2679.49   628.8 2681.72
#Mann= 6 ,-1,0
       0     .08       0      30      .1       0  327.07    .045       0
  393.58     .06       0     510      .1       0     570     .08       0
Bank Sta=327.07,393.58
XS Rating Curve= 0 ,0
Exp/Cntr=0.3,0.1

Type RM Length L Ch R = 1 ,7772    ,451.8,452.9,454.3
XS GIS Cut Line= 2
2200339.73248131575961.668750664 2199953.9969476 576547.09090286
#Sta/Elev= 30
       0 2692.02    23.4 2685.02    94.6 2636.56   104.8 2631.22   123.5 2623.16
   151.9 2617.89   166.4  2613.3   239.1 2612.41   262.1 2614.31   273.6 2612.67
   285.2 2613.86   296.4 2612.35   363.5 2612.47   411.4 2610.28   464.1 2612.38
   473.6 2609.05  503.822605.697   521.5 2604.38   540.7 2604.44  545.442605.698
   555.1 2611.36   573.5 2608.04   588.6 2608.32   597.1 2610.04   612.6 2625.48
   617.4    2629   631.7 2644.07   651.9 2661.95   672.1 2674.81   701.1  2689.5
#Mann= 4 ,-1,0
       0      .1       0  503.82    .045       0  545.44     .06       0
     640      .1       0
Bank Sta=503.82,545.44
XS Rating Curve= 0 ,0
Exp/Cntr=0.3,0.1

Type RM Length L Ch R = 1 ,7319    ,388.9,393.2,397.5
XS GIS Cut Line= 3
2199921.27483544575685.5773591422199898.55258846575849.971035035
2199572.95494259576282.364548723
#Sta/Elev= 30
       0 2660.74    35.9 2653.42   104.6 2646.84   112.7 2644.66     149    2630
   169.9 2623.38   189.9 2619.88   235.1 2616.31   280.1 2606.79   320.2 2603.15
   335.2 2604.94   372.7 2603.27   455.4  2604.1   478.4 2600.17  482.982598.292
     487  2596.8     509 2596.52   521.3 2596.71  526.042598.287   535.5 2606.21
   540.5 2607.56   558.4 2603.32   572.7 2603.59   580.6 2605.79   585.6 2609.21
   595.6  2619.6   600.6 2622.51   620.6 2627.99   650.7 2640.55   707.2 2678.99
#Mann= 6 ,-1,0
       0      .1       0     120     .08       0  475.96     .06       0
  482.98    .045       0  526.04     .06       0  605.96      .1       0
Bank Sta=482.98,526.04
XS Rating Curve= 0 ,0
Exp/Cntr=0.3,0.1

Type RM Length L Ch R = 1 ,6926    ,379.5,373.4,365.4
XS GIS Cut Line= 4
2199658.68887783575539.1358678242199573.75054106575703.270142186
2199283.02503268575969.9912816672199243.23554106576066.131920225
#Sta/Elev= 30
       0    2667    40.3 2650.37    83.8 2645.57   110.4  2635.9   119.4 2629.48
   137.4 2629.98   164.4 2624.28     178  2617.2   187.6 2607.55   192.9 2604.87
   208.7 2602.24   217.2  2597.3   224.9 2595.32   255.2  2595.4     292 2591.83
   323.7 2596.59   374.1 2599.22     377 2599.06  387.492592.674   425.8 2591.04
  438.972592.659   463.8 2600.28   496.4 2595.39     544 2595.95   560.4 2599.61
   582.8  2600.3   608.5 2612.29   656.4 2643.91   670.5 2648.68   683.4 2649.41
#Mann= 7 ,-1,0
       0      .1       0      10     .08       0  214.81      .1       0
  387.49    .045       0  438.97      .1       0  474.81     .06       0
  609.35      .1       0
#XS Ineff= 2 , 0
          373.33 2606.24  462.11         2607.29
Permanent Ineff=
       F       F
Bank Sta=387.49,438.97
XS Rating Curve= 0 ,0
Exp/Cntr=0.3,0.1

Type RM Length L Ch R = 1 ,6553    ,418.2,419.2,420.8
XS GIS Cut Line= 2
 2199279.9809002575368.5705834532198999.67935649575816.325840449
#Sta/Elev= 30
       0  2670.9    52.5 2667.25    71.5 2668.36    90.4  2667.5   104.5 2662.09
   122.2 2647.25   133.8 2635.01   150.4 2622.22   177.3 2606.23   194.2 2597.34
   203.6 2594.37   225.8 2591.25   250.8 2591.67   283.9  2590.5  291.742586.521
   293.4  2585.6   321.6    2585   345.2 2585.38  352.212586.522   384.1 2590.89
   399.2 2589.64   425.4  2590.6   436.9 2596.95   444.2 2603.31   453.1 2613.37
   458.5 2616.97   477.4 2624.27   491.5 2631.39     514  2639.8   528.3 2647.06
#Mann= 6 ,-1,0
       0     .08       0      40      .1       0  291.74    .045       0
  352.21      .1       0     400     .06       0     510      .1       0
Bank Sta=291.74,352.21
XS Rating Curve= 0 ,0
Exp/Cntr=0.3,0.1

Type RM Length L Ch R = 1 ,6133    ,348.9,339.3,325.9
XS GIS Cut Line= 2
2198980.14963381575090.7348206862198638.72645689575588.184718235
#Sta/Elev= 30
       0 2675.73    17.5 2669.32    32.1 2662.66    51.5 2653.66    63.6 2646.46
    85.2 2628.71    98.9 2616.26   131.2 2592.83   142.7  2587.5   180.1 2586.79
   192.2 2587.67   246.3  2587.6   257.8 2586.62   279.5 2587.23   313.5 2584.36
     362 2585.59   367.1 2585.24  379.452579.355   400.8 2578.36   436.2 2578.57
  440.252579.354   449.3 2583.38   459.4 2582.36     493 2581.83   512.4 2586.12
   541.5 2600.71   565.7 2610.68   575.4 2616.88   585.8 2620.09   603.3 2628.04
#Mann= 5 ,-1,0
       0     .08       0      30      .1       0  379.45    .045       0
  440.25     .06       0     510      .1       0
Bank Sta=379.45,440.25
XS Rating Curve= 0 ,0
Exp/Cntr(USF)=0,0
Exp/Cntr=0.3,0.1

Type RM Length L Ch R = 1 ,5794    ,481.4,477.3,472.6
XS GIS Cut Line= 3
2198493.83823197574865.9041745662198486.28730674 575050.29898764
2198404.23169326575483.223162206
#Sta/Elev= 30
       0 2650.57    27.3 2640.86    39.4  2634.9    51.3 2626.14    63.3 2623.38
    83.3 2610.59   112.4 2602.34   167.4 2590.82   184.5 2578.31   191.6 2574.95
   207.8 2573.71   228.2 2574.84   243.6 2579.38   277.8 2581.72   293.3 2578.43
   338.1 2579.04   366.6 2575.17     387  2575.4   403.3 2578.02   411.4 2573.19
   426.6 2571.57  461.612573.195   480.6 2577.95   496.8 2575.25   524.2 2576.51
   531.1 2580.99   537.6 2587.43   545.7 2597.91   551.6 2601.82   625.2 2617.96
#Mann= 4 ,-1,0
       0      .1       0   411.4    .045       0  461.61     .06       0
  554.55      .1       0
#XS Ineff= 2 , 0
        261.6414    2580
Permanent Ineff=
       F       F
Bank Sta=411.4,461.61
XS Rating Curve= 0 ,0
Exp/Cntr=0.3,0.1

Type RM Length L Ch R = 1 ,5317    ,454.9,455.4,456.1
XS GIS Cut Line= 2
2197966.32817957574884.5553815122197964.97339653575427.419685904
#Sta/Elev= 30
       0 2616.39     6.5 2614.65    36.6 2613.95    52.6 2605.47    88.6 2598.92
   108.6 2591.12   142.8 2569.21   152.6 2564.62   164.6 2563.05   180.6 2566.21
   212.6  2565.5   240.6 2569.03   256.6 2566.36   272.6 2568.35   312.6 2567.45
   336.6 2569.49   344.6 2568.28  350.272564.912   371.4 2563.75  394.652564.875
   404.6 2572.38   412.6 2572.67   421.7 2569.23   452.6 2568.93   456.6 2570.83
   464.6 2577.48   476.6 2592.97   496.6  2610.4   519.8 2633.61   542.9 2651.03
#Mann= 5 ,-1,0
       0      .1       0  350.27    .045       0  394.65      .1       0
     430     .06       0     530      .1       0
Bank Sta=350.27,394.65
XS Rating Curve= 0 ,0
Exp/Cntr=0.3,0.1

Type RM Length L Ch R = 1 ,4861    ,388.3,404.4,414.8
XS GIS Cut Line= 2
2197523.18895761574903.2516832482197503.89625935575421.328077426
#Sta/Elev= 30
       0 2632.23      58 2617.13      74 2606.51      90 2601.41     106 2593.79
     126 2579.74     146 2576.64     166  2560.9     174 2557.94   206.1 2555.57
   231.7 2559.15   266.1 2559.88   278.1 2563.15   298.1 2560.44   326.2 2561.39
   330.2 2560.36  335.342556.502   340.5 2554.88   358.2 2554.59  370.212556.536
   382.2 2564.51     410 2566.11   421.5 2571.93   434.2 2581.84   446.2 2595.46
   456.3 2604.78   466.3 2620.21   478.3 2631.44   502.3 2658.93   518.4 2670.62
#Mann= 5 ,-1,0
       0      .1       0     310     .06       0  335.34    .045       0
  370.21     .06       0     410      .1       0
Bank Sta=335.34,370.21
XS Rating Curve= 0 ,0
Exp/Cntr=0.3,0.1

Type RM Length L Ch R = 1 ,4457    ,351.4,345.6,341.1
XS GIS Cut Line= 4
2197239.37353371 574839.232074772197211.89632911575040.454571093
2197050.92512339575246.7615413192197035.35418693575345.853708274
#Sta/Elev= 30
       0 2621.16    22.3  2620.2    62.5 2616.31    82.7 2605.13    90.8  2602.3
   102.9 2600.12   132.4 2585.27   171.5 2574.64   199.8 2562.72   209.1 2557.02
   214.2 2555.34   280.4 2551.87   295.3 2549.53   305.5 2550.06   330.8 2549.22
  352.932550.075   371.6 2552.14   380.1 2556.34   384.7 2557.39   397.2 2554.21
   432.3 2554.33   451.3 2557.49   457.7 2559.52   462.8 2562.66   475.3 2574.19
   487.5  2583.3   507.7 2602.47   519.9 2610.34   544.1  2628.8   565.1 2646.59
#Mann= 5 ,-1,0
       0      .1       0   305.5    .045       0  352.93      .1       0
  393.09     .06       0  534.77      .1       0
Bank Sta=305.5,352.93
XS Rating Curve= 0 ,0
Exp/Cntr=0.3,0.1

Type RM Length L Ch R = 1 ,4111    ,188,184.7,174.7
XS GIS Cut Line= 2
2196964.65152492574696.0789979072196703.99512104575241.254715885
#Sta/Elev= 30
       0 2623.97    54.4 2605.62      81 2599.76   112.2 2595.08   130.9 2593.47
   143.1 2590.16   156.4 2589.88   214.2 2579.99   226.1 2574.88   249.5 2568.64
   267.2 2561.48   280.5 2554.03  292.312544.998   295.1 2543.87   302.7 2543.36
   342.6 2543.52  346.362544.986   353.5 2547.64   386.9 2547.25   409.1 2545.34
   422.4 2546.87   446.2 2544.74   460.1 2547.77   506.7 2547.89   511.1  2550.2
   517.1 2555.37   524.4 2559.15   557.5 2581.19     582 2599.74   604.3  2614.5
#Mann= 7 ,-1,0
       0      .1       0  292.31    .045       0  346.36      .1       0
     360     .06       0     390      .1       0     470     .06       0
     570      .1       0
Bank Sta=292.31,346.36
XS Rating Curve= 0 ,0
Exp/Cntr(USF)=0,0
Exp/Cntr=0.3,0.1

Type RM Length L Ch R = 1 ,3927    ,656.7,667.6,683.6
XS GIS Cut Line= 3
2196797.06459912574621.6747559672196667.78199224574864.729148659
2196593.58027348575240.525978886
#Sta/Elev= 30
       0 2620.72    26.6 2607.43    44.7 2600.78    85.5 2580.88    99.1 2576.54
   117.2  2573.7   135.4 2565.76   167.1 2556.59   195.5 2553.38   222.1 2546.09
     288 2545.82   300.2 2541.99   312.8 2541.51   333.2 2541.05  363.58 2541.53
   373.6 2544.31   434.8 2542.58   459.2 2546.96   471.5 2545.17     500 2544.81
   512.2 2546.57   516.3 2548.66   540.5 2568.78   548.9 2573.86   561.2 2586.13
   581.5 2599.34   601.9 2607.35   618.2 2610.49   634.6 2617.32   658.4 2631.95
#Mann= 5 ,-1,0
       0      .1       0   312.8    .045       0  363.58      .1       0
   435.3     .06       0   615.3      .1       0
#XS Ineff= 2 , 0
                          458.78         2550.94
Permanent Ineff=
       F       F
Bank Sta=312.8,363.58
XS Rating Curve= 0 ,0
Exp/Cntr=0.3,0.1

Type RM Length L Ch R = 1 ,3259    ,287.8,292.6,293.4
XS GIS Cut Line= 3
2196479.51771003574379.7094398422195985.97215813574962.749321893
2196097.61756487575235.500309839
#Sta/Elev= 30
       0  2629.7    33.4  2609.6    57.3 2587.05      80 2568.11    94.2 2557.88
   117.2 2545.02   141.4 2536.07   179.4 2537.82   185.1 2536.06   193.6  2529.6
   203.3 2528.68   227.3 2529.59   295.4 2532.73   342.6 2539.06   426.2 2537.31
   436.9 2535.55   478.8 2539.11   496.1 2534.79   511.4 2533.75   557.4 2541.88
   599.5 2541.85     642 2547.83   763.9 2557.67   805.4 2559.07   822.7 2563.17
   909.1 2604.36   935.1 2613.87   998.5 2628.78  1043.5 2644.07  1058.6 2651.21
#Mann= 5 ,-1,0
       0      .1       0   193.6    .045       0   227.3      .1       0
     450     .06       0     710      .1       0
#XS Ineff= 2 , 0
                          343.96         2544.98
Permanent Ineff=
       F       F
Bank Sta=193.6,227.3
XS Rating Curve= 0 ,0
Exp/Cntr=0.3,0.1

Type RM Length L Ch R = 1 ,2966    ,451.1,450.4,449.7
XS GIS Cut Line= 2
2196268.63173657574174.4494556222195666.55215577574934.391365529
#Sta/Elev= 30
       0 2663.82    23.9 2656.94    52.3 2645.45    67.8 2632.78    90.5 2608.91
   123.1 2582.14   190.2 2543.51   204.4 2532.83   224.4 2532.29  249.642525.348
   314.8 2524.15  322.182525.347   330.1 2532.76   335.4 2535.05   355.6  2535.3
   372.4 2532.65   437.3  2533.3   472.1 2529.33   488.3 2533.17   580.1 2537.57
   594.5 2534.11   619.1 2534.11   637.2 2539.21   702.6 2543.01   857.4 2545.09
   876.4 2551.99   913.4    2582   942.5 2582.92   962.9 2605.65   969.5 2610.72
#Mann= 5 ,-1,0
       0      .1       0  249.64    .045       0  322.18      .1       0
     570     .06       0     700      .1       0
Bank Sta=249.64,322.18
XS Rating Curve= 0 ,0
Exp/Cntr(USF)=0,0
Exp/Cntr=0.3,0.1

Type RM Length L Ch R = 1 ,2516    ,260.4,264.4,266.4
XS GIS Cut Line= 3
2195920.79695526573969.4567406542195758.64624699574094.404421553
2195321.15526701574652.554703269
#Sta/Elev= 30
       0 2673.57      21 2663.49    45.9 2646.44    54.4 2638.79    68.7 2636.06
     111 2605.73   152.3 2584.11   156.8 2580.48   182.8 2551.05   208.7  2527.2
   214.1 2523.29  230.26  2517.9   248.9 2516.22  280.572517.899   289.5 2525.21
   304.8 2526.19   325.3 2525.77   345.5 2522.13   401.4 2524.91   427.8 2523.24
   538.6 2527.56   574.2 2525.13   593.1  2528.5   778.3 2526.97   787.6 2530.17
   797.8 2537.36   831.2 2564.88   848.6 2583.91     858 2591.78   913.9 2606.89
#Mann= 5 ,-1,0
       0      .1       0  230.26    .045       0  280.57      .1       0
  504.71     .06       0  754.71      .1       0
Bank Sta=230.26,280.57
XS Rating Curve= 0 ,0
Exp/Cntr=0.3,0.1

Type RM Length L Ch R = 1 ,2252    ,121.2,113.1,98.8
XS GIS Cut Line= 4
 2195803.3094211573793.2189090762195639.94026656573848.287163417
2195219.58592509574281.4907642342195111.28502488574329.216584663
#Sta/Elev= 30
       0 2655.98      16  2642.5    28.6  2640.6    62.5 2615.86    83.5 2603.98
   147.7 2562.83   183.6 2531.51   195.9 2522.85   209.6 2519.23     286 2519.97
   298.4 2514.53   327.2 2512.95   351.1 2513.12  357.152514.545   401.8 2522.59
   436.3 2517.95   458.6 2519.82   523.6 2521.08   636.3 2517.17   647.4 2519.16
     689 2520.01   769.7 2525.35   792.9 2530.63   811.8 2538.69   819.1 2543.33
   832.2 2554.42   840.9 2556.32   848.2 2560.22   863.3 2574.17   894.4 2587.99
#Mann= 4 ,-1,0
       0      .1       0   298.4    .045       0  357.15     .06       0
   492.4      .1       0
#XS Ineff= 2 , 0
                          398.53         2531.96
Permanent Ineff=
       F       F
Bank Sta=298.4,357.15
XS Rating Curve= 0 ,0
Exp/Cntr(USF)=0,0
Exp/Cntr=0.3,0.1
